HEC-RAS study Crooked_Creek.prj: Crooked_Creek

--- Crooked_Creek.g05 (geometry) --- (continued)

Type RM Length L Ch R = 1 ,58388.72,338.89,329.93,311.12
XS GIS Cut Line= 3
  1053777.783449   680496.851306  1054265.004872   680196.051798
  1054766.306963   679967.709209
#Sta/Elev= 30
       0 1498.63   58.93 1493.07   91.14 1487.99  123.78 1485.51  139.77 1481.33
  173.29 1479.98  189.07 1474.24  205.26 1472.34  276.54 1466.29  365.82 1463.82
  413.15 1463.82  430.98 1464.99  497.96  1462.6  549.13 1463.91  562.33 1458.46
  572.59 1456.79  589.53 1460.82  631.29 1467.12  655.61 1481.14  700.99 1504.52
  721.34 1516.25  777.46 1544.88  851.52 1576.75  904.62  1593.6  967.86 1610.77
 1045.25 1635.57 1059.89 1644.25 1065.54 1646.36 1093.34  1651.7 1123.45 1652.93
#Mann= 3 , 0 , 0
       0      .1       0  549.13    .045       0  589.53      .1       0
Bank Sta=549.13,589.53
Exp/Cntr=0.3,0.1

Type RM Length L Ch R = 1 ,58058.79,371.21,364.69,357.19
XS GIS Cut Line= 2
  1053968.068085   680935.976136  1054729.944635   680159.656421
#Sta/Elev= 30
       0 1560.65   28.01 1557.85   71.45 1551.24   94.26 1544.94  131.16 1537.21
  167.33 1528.16  231.31 1508.76   244.1    1503  256.77 1498.84  268.72 1493.15
  283.25 1488.34  291.27 1488.39   314.5  1484.9  334.46 1480.92  347.36  1475.9
  373.23 1475.93  403.06 1470.37  431.87 1468.22  587.28 1462.13  653.95 1461.22
     669 1461.98  687.76 1455.59  713.34 1462.97   731.3 1465.55  744.19 1470.57
   781.1 1494.49  919.68 1576.75 1019.36 1617.72 1043.42 1628.69 1087.72 1644.25
#Mann= 3 , 0 , 0
       0     .07       0     669    .045       0  713.34      .1       0
Bank Sta=669,713.34
Exp/Cntr=0.3,0.1

Type RM Length L Ch R = 1 ,57694.1 ,532.67,542.64,552.42
XS GIS Cut Line= 3
  1054313.100416   681162.832233  1054654.105865   680747.316054
  1054993.389902   680261.910377
#Sta/Elev= 30
       0 1550.44   103.4 1536.86   144.8 1529.84  200.35 1518.11  243.77 1504.74
  270.46 1493.78  297.62 1479.97  313.97 1475.83  337.67  1475.3  352.44 1471.18
  392.66 1466.78  451.58 1462.91  509.29 1460.77  541.44 1461.45  563.12  1459.4
   585.8 1454.77  607.48 1459.67  666.96 1462.85  677.16 1466.99  713.94 1488.54
  719.18 1493.09  784.74 1528.88  802.14 1534.59     863 1561.12  893.37 1566.08
  933.16 1579.98 1028.61  1608.3 1047.98 1615.82  1095.2 1642.42 1129.76 1655.57
#Mann= 3 , 0 , 0
       0      .1       0  563.12    .045       0  607.48      .1       0
Bank Sta=563.12,607.48
Exp/Cntr=0.3,0.1

Type RM Length L Ch R = 1 ,57151.46,534.01,562.75,584.3
XS GIS Cut Line= 3
  1054694.294214   681285.397651  1055249.898293   680777.101402
  1055567.647723   680495.459845
#Sta/Elev= 30
       0 1529.55    4.29 1528.46   22.98 1519.34   42.52 1515.55   73.74 1504.22
   86.74 1502.53  122.62 1488.51  153.16 1487.31  168.71 1477.23  185.13 1472.39
  210.19 1472.12  229.09 1467.34  383.95 1459.81  476.59 1461.09  646.74 1459.66
  673.49 1455.81  686.45  1452.2  695.28 1453.57  710.07 1459.27  775.26 1471.57
  799.42 1478.59  837.63 1485.07  909.11 1504.42  961.75 1515.81 1029.77 1537.52
 1082.47    1553 1118.17 1566.48 1151.63 1581.48 1171.07 1591.51 1177.64 1593.62
#Mann= 3 , 0 , 0
       0     .07       0  646.74    .045       0  710.07      .1       0
Bank Sta=646.74,710.07
Exp/Cntr=0.3,0.1

Type RM Length L Ch R = 1 ,56588.72,285.58,260.97,234.95
XS GIS Cut Line= 3
  1054758.603618   681420.187136   1055282.96048   681314.793511
  1055780.480823    681180.05459
#Sta/Elev= 30
       0 1545.93   13.09 1544.51   34.35 1545.26   76.64 1540.21  167.25 1520.34
   203.4 1508.13  235.57 1493.21  243.04 1486.86  262.65 1466.11  264.02 1465.67
   296.4 1467.44  312.34 1463.23  328.75 1461.06  458.81 1459.01   513.9 1456.69
  534.84 1450.31  560.66 1453.37  571.99 1456.52  582.03 1459.74  601.47 1462.65
  630.26 1474.64  643.23 1482.21  683.86 1497.34  746.31 1508.19  844.61  1512.3
  938.49 1524.91  954.61 1528.94  982.67  1539.4 1015.06 1549.39 1050.29    1558
#Mann= 3 , 0 , 0
       0     .07       0   513.9    .045       0  571.99      .1       0
Bank Sta=513.9,571.99
Exp/Cntr=0.3,0.1

Type RM Length L Ch R = 1 ,56327.75,40.69,43.05,42.88
XS GIS Cut Line= 4
  1054758.866888   681964.239791  1055339.427234   681577.156258
  1055373.763868    681555.94834  1055669.702138   681275.520025
#Sta/Elev= 30
       0 1533.62   48.22 1522.61   79.09 1514.35   96.12 1511.76  144.45 1497.34
  163.47 1493.79  210.43 1482.39  254.21 1473.65  286.23 1470.31  334.65 1466.24
     409 1465.01  437.58 1466.06  469.87 1462.99  502.51 1461.24  679.32 1457.37
  757.41 1457.77   773.4 1452.34  778.95 1449.33  791.78  1450.8  810.41 1455.46
  819.42 1456.38   830.7 1457.63  875.58 1458.21  882.71  1460.1  922.02 1487.07
  950.29 1504.19  998.36 1524.33 1012.32 1527.88 1052.08 1533.83 1145.83 1541.64
#Mann= 3 , 0 , 0
       0     .07       0  757.41    .045       0  819.42      .1       0
Bank Sta=757.41,819.42
Exp/Cntr=0.5,0.3

Type RM Length L Ch R = 1 ,56284.7 ,40.7,43.34,43.3
BEGIN DESCRIPTION:
Upstream xs of Bridge 37111-0249
END DESCRIPTION:
XS GIS Cut Line= 4
  1054781.056622   681997.520664  1055361.038504   681610.822813
  1055398.287577   681587.816005  1055697.215338   681304.554903
#Sta/Elev= 30
       0  1520.5    27.5  1513.9    82.4  1504.1    95.3  1500.6   113.7    1498
   126.3  1494.8   187.9  1483.7   270.3  1471.7   304.4  1468.5   389.4  1464.8
   422.2  1466.5   485.3    1462   721.9  1457.9   742.3  1456.8   757.9  1452.7
   760.9  1448.4   766.9    1447   778.9  1448.4   783.6    1453   785.7  1453.1
   816.9  1458.2   873.7  1456.6   888.3  1459.2   955.3  1502.4  1007.4  1525.8
  1041.6  1533.6  1056.7  1541.5  1064.7  1543.2  1093.4  1547.8  1152.7    1555
#Mann= 3 , 0 , 0
       0     .07       0   757.9    .045       0   785.7      .1       0
#XS Ineff= 2 , 0
       0   732.7  1458.7   807.1       0  1457.5
Permanent Ineff=
       F       F
Bank Sta=757.9,785.7
Exp/Cntr=0.5,0.3

Type RM Length L Ch R = 3 ,56263.02,,,
BEGIN DESCRIPTION:
Bridge : 37111-0249,  Private Dr.
END DESCRIPTION:
Bridge Culvert--1,0,-1,-1, 0
Deck Dist Width WeirC Skew NumUp NumDn MinLoCord MaxHiCord MaxSubmerge Is_Ogee
15.2,13,2.6,0, 52, 49, , , 0.95, 0, 0,0,,
   490.4   492.3   506.3     510   522.4     528   538.9   546.3   555.2   564.2
   571.3   582.4   587.7   600.9   604.3   619.5     621   634.2   637.4     638
   653.3   656.7   669.6   675.5   685.4     694   696.7   699.7   702.4   715.6
   722.1   729.3   742.2   747.9   747.9   791.9   791.9   802.4   817.2   826.6
   833.2   841.3   846.3   856.2   868.6   871.3   876.9   886.6     897   902.1
   917.2   925.7
  1461.5  1461.5  1461.3  1461.3  1461.1    1461  1460.8  1460.3  1460.2    1460
  1459.9  1459.8  1459.7  1459.3  1459.2  1459.1    1459    1459    1459    1459
    1459  1458.8  1458.8  1458.8  1458.8  1458.8  1458.8  1458.8  1458.8  1458.8
  1458.8  1458.8  1458.8  1458.8  1458.8  1458.8  1458.8  1458.8  1458.8  1457.6
  1457.5  1457.5  1457.5  1457.8  1458.6  1458.8  1459.4  1459.7  1462.6  1463.9
  1474.2  1479.1
                                                                                
                                                                                
                                                                                
                                  1455.1  1455.1
                                                                                
                
   461.8   506.3     510   522.4     528   538.9   546.3   555.2   564.2   571.3
   582.4   587.7   600.9   604.3   619.5     621   634.2   637.4     638   653.3
   656.7   669.6   675.5   685.4     694   696.7   699.7   702.4   715.6   722.1
   729.3   742.2     746     746     790     790   802.4   817.2   826.6   833.2
   841.3   846.3   856.2   868.6   871.3   876.9   886.6     897   902.1
  1461.9  1461.3  1461.3  1461.1    1461  1460.8  1460.3  1460.2    1460  1459.9
  1459.8  1459.7  1459.3  1459.2  1459.1    1459  1458.8  1458.8  1458.8  1458.8
  1458.8  1458.8  1458.8  1458.8  1458.8  1458.8  1458.8  1458.8  1458.8  1458.8
  1458.8  1458.8  1458.8  1458.8  1458.8  1458.8  1458.8  1458.8  1457.6  1457.5
  1457.5  1457.5  1457.8  1458.6  1458.8  1459.4  1459.7  1462.6  1463.9
                                                                                
                                                                                
                                                                                
                          1455.1  1455.1
                                                                        
BR Coef=-1 , 1 , 0 ,, 0 ,,,0.8,0,1.2,0,
WSPro=,,,, 1 ,,,, 0 ,,,, 0 ,,,,-1 ,-1 ,-1 , 0 , 0 , 0 , 0 , 0
BC Design=,, 0 ,, 0 ,,,,,,

Type RM Length L Ch R = 1 ,56241.35,40.03,41.58,42.44
BEGIN DESCRIPTION:
Down stream xs of Bridge 37111-0249
END DESCRIPTION:
XS GIS Cut Line= 4
  1054803.246357   682030.801537  1055382.649735   681644.489406
  1055422.811286   681619.683708  1055724.728498    681333.58982
#Sta/Elev= 30
       0  1511.2    72.6  1499.6   152.7  1490.3   270.2  1472.1   340.6  1466.3
   390.8  1464.9   409.3    1467   451.6  1462.7   481.7  1461.1   663.3  1457.5
   724.7  1457.7   749.8  1455.6  752.231454.463     756  1452.7     759  1448.4
     765    1447     777  1448.4  792.541455.703   808.6  1456.7   865.6  1456.6
   879.5  1458.4   912.8  1465.4   920.2  1469.6     961  1500.5  1021.7  1528.7
  1033.6  1533.3  1059.8  1541.1  1072.8  1548.5  1097.6  1554.4  1159.5  1566.7
#Mann= 3 , 0 , 0
       0     .07       0  752.23    .045       0  792.54      .1       0
#XS Ineff= 2 , 0
       0   730.9  1458.5   805.1       0  1457.4
Permanent Ineff=
       F       F
Bank Sta=752.23,792.54
Exp/Cntr=0.5,0.3

Type RM Length L Ch R = 1 ,56199.77,309.38,290.92,275.51
XS GIS Cut Line= 4
  1054825.436091    682064.08241  1055404.261004   681678.155961
  1055447.334996   681651.551372  1055752.241698   681362.624697
#Sta/Elev= 30
       0 1508.24   28.65 1505.68   75.63 1503.57      87 1501.84  138.27 1496.87
  186.18 1489.35   201.8 1485.56  263.52 1473.68  325.23 1466.05  389.19 1464.42
  405.64 1466.78  443.39 1462.18   485.1  1460.5  535.59 1460.28   613.1 1458.31
  729.19 1456.75  755.83 1448.84  761.18 1450.79  808.42 1456.67  886.17 1455.61
  922.04 1466.32  954.22 1486.11  972.78 1498.76 1004.65 1512.13 1018.46 1519.96
 1059.65 1541.07 1073.65 1549.08  1101.4 1559.36 1135.34 1567.79 1166.37 1574.25
#Mann= 3 , 0 , 0
       0     .07       0  729.19    .045       0  808.42      .1       0
Bank Sta=729.19,808.42
Exp/Cntr=0.3,0.1

Type RM Length L Ch R = 1 ,55908.85,496.93,520.13,529.81
XS GIS Cut Line= 3
  1055281.774074   682349.991943  1055722.011599   681711.215973
  1055976.026283   681247.044233
#Sta/Elev= 30
       0 1539.58   73.43 1517.64  111.05 1508.99  167.54 1492.09  184.01 1490.13
  257.76 1472.65  271.61 1468.04  292.87 1467.35  327.54 1461.19  382.36 1458.33
  520.13 1455.74  743.88 1455.95  759.58 1453.33  766.11 1448.65  806.98 1456.29
  820.47 1457.42  831.44 1460.16  837.99 1464.61  852.28 1469.54  869.05 1477.51
  933.34 1510.96  957.29 1520.58  993.33  1537.6 1024.18 1545.08 1046.83 1555.06
 1091.12 1564.79 1145.68 1588.66 1231.28  1597.5 1246.06 1601.03 1304.92 1608.74
#Mann= 3 , 0 , 0
       0      .1       0  743.88    .045       0  806.98      .1       0
Bank Sta=743.88,806.98
Exp/Cntr=0.3,0.1

Type RM Length L Ch R = 1 ,55388.72,457.67,462.58,468.39
XS GIS Cut Line= 3
  1055448.661522   682421.926204  1056044.425056   682013.505585
  1056352.155496   681774.518084
#Sta/Elev= 30
       0  1528.1   74.08 1513.72   83.86 1510.87   98.02 1502.93  108.33 1501.19
  159.65 1499.95   175.6 1496.88  191.06 1490.84  222.35 1484.36  237.73 1479.55
  253.87 1478.52   269.3 1467.66   313.4 1467.76  358.36 1457.78   557.8 1453.55
  712.11 1454.89  715.07 1451.52  722.32 1446.78  748.25 1455.61  802.98 1462.38
  816.31 1465.53  847.37 1478.53  883.44 1496.49  961.58 1542.75  988.97 1562.06
 1021.53 1577.67 1060.94 1599.28 1081.25 1604.48 1098.76 1611.76 1111.95 1611.69
#Mann= 3 , 0 , 0
       0      .1       0  712.11    .045       0  748.25      .1       0
Bank Sta=712.11,748.25
Exp/Cntr=0.3,0.1

Type RM Length L Ch R = 1 ,54926.14,476.63,486.27,409.8
XS GIS Cut Line= 3
  1055592.529967    682752.82369  1056116.211196   682433.435686
  1056637.015055   682062.255013
#Sta/Elev= 30
       0 1561.03   27.65 1565.77   60.24 1568.36   78.62 1566.92  106.98 1561.54
  176.43 1539.41  242.57  1512.5  288.54 1499.52  334.42 1483.81  349.58 1477.81
  363.66 1466.59  395.82 1466.28  411.44 1460.93  443.87 1457.63  514.95 1456.35
  542.82  1453.5  557.35 1445.43   574.2 1450.51  635.28 1452.82  808.86 1452.91
  897.82 1454.78  914.41 1462.41  973.46 1497.95  1026.8 1526.39 1088.91 1554.16
 1123.48 1573.82 1139.87 1579.41 1188.46 1589.95 1220.49 1599.23 1252.93 1603.11
#Mann= 3 , 0 , 0
       0     .07       0  542.82    .045       0   574.2     .07       0
Bank Sta=542.82,574.2
Exp/Cntr=0.3,0.1

Type RM Length L Ch R = 1 ,54439.88,46.12,46.28,47.58
XS GIS Cut Line= 6
  1055872.860687     682985.6924  1056239.239774   682890.016395
  1056315.071516   682792.732302  1056360.010846   682682.452429
  1056421.798658   682618.140888  1056680.037705   682139.211294
#Sta/Elev= 30
       0 1509.91   47.76 1505.58  108.45 1498.12  158.51 1489.65  173.99 1488.11
  189.12 1484.49  238.95 1477.63  298.29  1467.2  317.64 1462.48  372.61 1460.81
  405.39 1455.78  647.45 1453.51  689.27 1450.63  703.91 1448.09   708.9  1443.6
  723.31 1443.83  741.37 1451.19  870.53 1452.97  906.75  1452.4  919.96  1454.2
  972.78  1478.9  988.31  1487.2    1007 1493.57 1040.54 1510.24 1078.39 1533.39
 1109.77 1555.06 1159.58 1593.24 1178.63 1604.26 1197.02 1609.42  1254.4    1616
#Mann= 3 , 0 , 0
       0     .07       0  689.27    .045       0  741.37     .07       0
Bank Sta=689.27,741.37
Exp/Cntr=0.5,0.3

Type RM Length L Ch R = 1 ,54393.59,55.47,55.66,58.06
BEGIN DESCRIPTION:
Upstream xs of Bridge 37111-0333
END DESCRIPTION:
XS GIS Cut Line= 6
   1055884.23067   683029.232309  1056265.359378   682929.704612
  1056354.393158   682815.483646  1056398.431528   682707.414753
  1056458.497306   682644.895618  1056719.646696   682160.568498
#Sta/Elev= 30
       0  1507.7   138.2  1497.7   190.8    1491     221  1482.4     313  1478.1
   333.6  1471.4   361.1  1464.9     380  1461.7     413  1459.8   433.1  1456.7
   625.1    1454   686.6  1451.9   697.1  1452.6  713.431450.484     718  1448.1
     724  1442.2     733  1441.9  755.991450.296   946.1  1452.4   967.8  1457.8
   981.8    1467  1006.6  1479.6  1052.4  1500.8  1088.7  1514.9  1109.5  1527.1
  1120.1  1531.7  1145.5  1547.1  1188.6  1580.5  1227.9  1607.3  1292.4  1620.5
#Mann= 3 , 0 , 0
       0     .07       0  713.43    .045       0  755.99     .07       0
#XS Ineff= 2 , 0
       0   688.9  1453.3   769.1       0    1451
Permanent Ineff=
       F       F
Bank Sta=713.43,755.99
Exp/Cntr=0.5,0.3

Type RM Length L Ch R = 3 ,54363.48,,,
BEGIN DESCRIPTION:
Bridge : 37111-0333,  Private Dr.
END DESCRIPTION:
Bridge Culvert--1,0,-1,-1, 0
Deck Dist Width WeirC Skew NumUp NumDn MinLoCord MaxHiCord MaxSubmerge Is_Ogee
24.1,12,2.6,0, 47, 59, , , 0.95, 0, 0,0,,
   606.1   612.7     621   624.2   634.3   643.1   645.8   651.4   653.6   654.7
     660   664.9   672.1   677.8   690.7     691   691.7   710.5   712.2     713
     713     745     745   745.1   753.1   757.7   765.2   765.9   766.3   778.8
   786.3   791.2     800   801.8   863.6   873.1   874.7   876.6   886.1   894.5
   898.8   909.3     914   931.9   933.2   947.4   948.3
  1454.1    1454  1453.8  1453.8  1453.7  1453.8  1453.8  1453.4  1453.4  1453.4
  1453.4  1453.4  1453.4  1453.4  1453.4  1453.4  1453.4  1453.4  1453.4  1453.4
  1453.4  1453.4  1453.4  1453.4  1453.4  1452.3    1452    1452    1452  1451.8
  1451.6  1451.6  1451.1    1451  1451.5    1452    1452    1452  1451.8  1451.8
    1452  1452.2    1452  1452.1  1452.1  1452.6  1452.7
                                                                                
                                                                                
  1450.6  1450.6
                                                                                
                                                        
   496.5   497.1   497.8   512.3   524.9   528.3   532.3   539.7   547.8   549.3
   550.7   562.6   570.4   576.5   582.8   584.8   589.9   597.6   601.9   607.9
   613.3   617.4   627.7     631     644   650.5   658.8     662   672.2   680.9
   683.7   689.2   691.4   692.5   697.9   702.8     710   715.7   728.5   728.8
   729.6   748.4     749     749     781     781   782.9   790.9   795.5     803
   803.8   804.2   816.6   824.1     829   837.9   839.7   971.1     997
  1456.9  1456.8  1456.8  1456.3  1455.9  1455.8  1455.7  1455.5  1455.6  1455.5
  1455.5  1455.3  1455.3  1455.3  1455.1  1455.1  1454.9  1454.8  1454.7  1454.6
  1454.5  1454.5  1454.3  1454.2  1454.1    1454  1453.8  1453.8  1453.7  1453.8
  1453.8  1453.4  1453.2  1453.3  1453.5  1453.4  1453.4  1453.4  1453.4  1453.4
  1453.4  1453.4  1453.4  1453.4  1453.4  1453.4  1453.4  1453.4  1452.3    1452
    1452    1452  1451.8  1451.6  1451.6  1451.1    1451  1452.1  1453.1
                                                                                
                                                                                
                                                                                
                                                                                
                          1450.6  1450.6
                                                                        
BR Coef=-1 , 1 , 0 ,, 0 ,,,0.8,0,1.2,0,
WSPro=,,,, 1 ,,,, 0 ,,,, 0 ,,,,-1 ,-1 ,-1 , 0 , 0 , 0 , 0 , 0
BC Design=,, 0 ,, 0 ,,,,,,

Type RM Length L Ch R = 1 ,54337.93,99.56,81.59,67.29
BEGIN DESCRIPTION:
Down stream xs of Bridge 37111-0333
END DESCRIPTION:
XS GIS Cut Line= 6
  1055898.127332   683082.447739  1056297.283315   682978.212402
  1056402.452973   682843.290874  1056445.390105   682737.924279
  1056503.351158   682677.595813  1056768.057667   682186.671712
#Sta/Elev= 30
       0  1499.1     100  1492.6   208.3  1479.8   284.4  1478.1   365.1    1463
   378.1    1462     430  1461.7   519.2  1456.6   524.1  1455.1   700.6  1453.6
  745.381450.903     754  1448.1     760  1442.2     769  1441.9  790.071451.284
   974.6  1452.1  1004.1  1454.1  1016.4  1458.1  1032.7  1469.8  1090.7  1499.4
  1130.8  1513.1  1172.2  1529.9  1184.4  1536.6  1200.3    1552  1218.8  1563.2
  1245.6  1575.7  1263.6  1589.1  1286.6  1603.6    1309  1611.6  1338.8  1618.5
#Mann= 3 , 0 , 0
       0     .08       0  745.38    .045       0  790.07     .07       0
#XS Ineff= 2 , 0
       0   729.4  1453.4   800.6       0  1450.8
Permanent Ineff=
       F       F
Bank Sta=745.38,790.07
Exp/Cntr=0.5,0.3

Type RM Length L Ch R = 1 ,54256.34,561.7,587.01,596.43
XS GIS Cut Line= 3
  1056252.077103   683431.254711  1056550.950804   682713.181534
  1056807.666658   682208.028877
#Sta/Elev= 30
       0 1514.54   68.85 1502.42  118.17 1496.51  155.38 1488.69  177.91 1487.49
  307.82 1468.82  348.22  1467.4  375.32 1464.09  395.83 1464.74  422.07 1463.09
  472.21 1455.97  553.06 1454.04  663.68 1453.96  703.16 1451.81  712.24 1447.33
  727.03 1443.11  751.95 1445.35  763.43 1451.06  994.46 1452.37 1011.46 1454.59
 1078.27 1488.89 1110.22 1502.15 1148.89  1514.1 1181.04 1527.53 1208.68 1548.41
 1243.58 1567.12 1272.71 1587.16 1295.74 1599.46 1325.44 1609.71 1344.43    1614
#Mann= 3 , 0 , 0
       0     .08       0  703.16    .045       0  763.43     .07       0
Bank Sta=703.16,763.43
Exp/Cntr=0.3,0.1

Type RM Length L Ch R = 1 ,53669.32,45.8,48.44,47.77
XS GIS Cut Line= 4
  1056597.222991    683581.58922  1056814.930028   683176.316776
  1056858.922145   683137.893297  1057274.344883   682541.906572
#Sta/Elev= 30
       0 1504.98   69.45 1497.84   116.9 1491.54  128.18 1491.53  196.16 1485.62
  287.03 1475.93  298.56 1473.69  329.63 1473.69  347.66  1468.3   399.1 1461.47
  432.03 1458.24  465.43  1456.3  496.08 1449.28  512.69 1447.97  529.92 1441.45
  561.15 1448.23  587.78 1450.06  658.91 1449.75   717.7 1450.65  813.71 1449.01
     957 1451.67 1039.67 1454.88 1068.64 1458.45 1102.28 1470.66 1121.05 1475.98
 1132.36 1482.41 1150.26 1488.76  1222.9 1505.64 1234.94 1509.74 1244.94 1514.65
#Mann= 3 , 0 , 0
       0     .08       0  512.69    .045       0  561.15     .07       0
Bank Sta=512.69,561.15
Exp/Cntr=0.5,0.3

Type RM Length L Ch R = 1 ,53620.89,83.47,61.81,65.29
BEGIN DESCRIPTION:
Upstream xs of Bridge 37111-0334
END DESCRIPTION:
XS GIS Cut Line= 4
  1056636.865264   683602.884519  1056850.698201   683204.823948
  1056892.682256   683168.154349  1057311.261713   682567.638862
#Sta/Elev= 30
       0  1509.9   109.8  1495.4   151.1  1491.7   203.3  1489.2   231.3  1482.7
   282.8  1478.1   293.4  1473.7   329.8  1472.5   355.1  1468.6   379.1  1466.5
   428.3  1458.2   469.1  1455.2  487.51 1447.01     502  1442.1     504  1440.5
     522  1441.3   530.5    1447   544.1  1450.8   626.5  1449.2   689.2  1450.3
   803.1  1449.1   946.2  1451.4  1055.3  1455.3  1081.6  1458.8  1127.6  1475.5
  1173.8  1484.9  1189.8  1490.3  1209.5  1494.9  1221.1  1499.2  1239.6  1508.5
#Mann= 3 , 0 , 0
       0     .08       0  487.51    .045       0   530.5     .07       0
#XS Ineff= 2 , 0
       0   463.6  1451.4   552.4       0  1449.2
Permanent Ineff=
       F       F
Bank Sta=487.51,530.5
Exp/Cntr=0.5,0.3

Type RM Length L Ch R = 3 ,53590.45,,,
BEGIN DESCRIPTION:
Bridge : 37111-0334, Paved Private Dr.
END DESCRIPTION:
Bridge Culvert--1,0,-1,-1, 0
Deck Dist Width WeirC Skew NumUp NumDn MinLoCord MaxHiCord MaxSubmerge Is_Ogee
24.4,12,2.6,0, 106, 93, , , 0.95, 0, 0,0,,
   344.2   345.4   358.3   361.1   367.9   375.1   392.3   394.5   404.4   407.6
     418   418.1   418.2   430.3   442.2   443.5   456.4   458.6   460.3   460.7
   475.2   477.2   480.9   483.5     488     488     528     528   539.3   543.9
   561.8   565.2   569.5   574.2   576.7   585.8   593.6   598.3   603.8   611.9
   620.8   627.2   640.5   644.5   646.5   661.8   662.6   675.7   685.8   687.9
   691.2   695.5   698.1   704.9   711.6   715.5   719.5   725.8   733.8   736.8
     744   754.6   759.1   768.8   777.8   782.3   790.3   797.5   801.6     811
   819.4     824   828.2   837.7   848.2   850.5   852.6   867.8   870.1   871.9
   883.4   895.5   896.8   898.4   908.3   919.1   919.5     920   930.8   937.9
   942.1   948.7   953.9   962.2   965.8   968.1   981.3   996.3   997.8  1002.5
  1012.9  1016.4  1028.1  1040.9  1043.1  1045.2
  1471.3  1471.2  1469.8  1469.5  1469.1  1468.9  1467.2    1467  1465.3  1464.7
  1462.9  1462.9  1462.9  1459.8  1459.2  1458.9  1456.9  1456.6  1456.5  1456.4
  1453.1  1452.3  1451.5  1451.5  1451.5  1451.5  1451.5  1451.5  1451.5  1451.5
  1450.6  1450.6  1450.3    1450    1450  1449.7  1449.9  1449.8  1449.7  1449.5
  1449.3  1449.1    1449    1449    1449  1449.1  1449.1  1449.6  1449.7  1449.7
  1449.7  1449.7  1449.7  1449.8  1449.7  1449.7  1449.6  1449.6  1449.5  1449.5
  1449.4  1449.2  1449.2    1449    1449  1448.9  1449.1  1449.2  1449.3  1449.5
  1449.6  1449.7  1449.8    1450  1450.1  1450.2  1450.2  1450.3  1450.3  1450.3
  1450.3  1450.4  1450.4  1450.5  1450.7  1450.9  1450.9  1450.9  1451.1  1451.2
  1451.3  1451.4  1451.5  1451.6  1451.7  1451.7  1452.1  1452.5  1452.6  1452.8
  1453.2  1453.3  1453.7  1454.2  1454.3  1454.4
                                                                                
                                                                                
                                          1448.8  1448.8
                                                                                
                                                                                
                                                                                
                                                                                
                                                                                
                                                                                
                                                                                
                                                
   372.6     383   383.1   383.2   395.3   407.2   408.5   421.4   423.6   425.3
   425.7   440.2   442.2   445.9   448.5     457     457     497     497   504.3
   508.9   526.8   530.2   534.5   539.2   541.7   550.8   558.6  563.29   568.8
   576.9   585.8   592.2   605.5   609.5   611.5   626.8   627.6   640.7   650.8
   652.9   656.2   660.5   663.1   669.9   676.6   680.5   684.5   690.8   698.8
   701.8     709   719.6   724.1   733.8   742.8   747.3   755.3   762.5   766.6
     776   784.4     789   793.2   802.7   813.2   815.5   817.6   832.8   835.1
   836.9   848.4   860.5   861.8   863.4   873.3   884.1   884.5     885   895.8
   902.9   907.1   913.7   918.9   927.2   930.8   933.1   946.3   961.3   962.8
   967.5   977.9   981.4
  1464.7  1462.9  1462.9  1462.9  1459.8  1459.2  1458.9  1456.9  1456.6  1456.5
  1456.4  1453.1  1452.3  1451.5  1451.5  1451.5  1451.5  1451.5  1451.5  1451.5
  1451.5  1450.6  1450.6  1450.3    1450    1450  1449.7  1449.9  1449.8  1449.7
  1449.5  1449.3  1449.1    1449    1449    1449  1449.1  1449.1  1449.6  1449.7
  1449.7  1449.7  1449.7  1449.7  1449.8  1449.7  1449.7  1449.6  1449.6  1449.5
  1449.5  1449.4  1449.2  1449.2    1449    1449  1448.9  1449.1  1449.2  1449.3
  1449.5  1449.6  1449.7  1449.8    1450  1450.1  1450.2  1450.2  1450.3  1450.3
  1450.3  1450.3  1450.4  1450.4  1450.5  1450.7  1450.9  1450.9  1450.9  1451.1
  1451.2  1451.3  1451.4  1451.5  1451.6  1451.7  1451.7  1452.1  1452.5  1452.6
  1452.8  1453.2  1453.3
                                                                                
                                                  1448.8  1448.8
                                                                                
                                                                                
                                                                                
                                                                                
                                                                                
                                                                                
                                                                                
                        
BR Coef=-1 , 1 , 0 ,, 0 ,,,0.8,0,1.2,0,
WSPro=,,,, 1 ,,,, 0 ,,,, 0 ,,,,-1 ,-1 ,-1 , 0 , 0 , 0 , 0 , 0
BC Design=,, 0 ,, 0 ,,,,,,

Type RM Length L Ch R = 1 ,53559.08,63.46,50.49,49.24
BEGIN DESCRIPTION:
Down stream xs of Bridge 37111-0334
END DESCRIPTION:
XS GIS Cut Line= 4
  1056689.721655    683631.27825  1056898.389073    683242.83351
  1056937.695685   683208.502391  1057360.484127   682601.948504
#Sta/Elev= 30
       0  1514.4    58.2  1506.7   132.6  1494.1   191.9  1487.5   242.4  1478.7
   277.4  1475.3   289.1  1471.3     314  1471.7   368.9  1467.7   403.1  1456.3
     425  1455.3   450.3  1449.9  451.42 1448.16  457.97 1444.43     473  1440.5
     491  1441.3     491  1442.1  498.07 1447.04  501.11  1450.2   519.5  1451.2
   611.7  1448.9   676.8  1449.7   752.2  1448.8   944.4  1451.6  1075.4  1456.8
  1093.5  1460.7  1113.4  1460.8    1126  1465.2  1172.2  1473.2  1232.5  1491.4
#Mann= 3 , 0 , 0
       0     .08       0  451.42    .045       0  498.07     .07       0
#XS Ineff= 2 , 0
       0   431.6  1454.9   522.4       0    1449
Permanent Ineff=
       F       F
Bank Sta=451.42,498.07
Exp/Cntr=0.5,0.3

Type RM Length L Ch R = 1 ,53508.59,605.87,603.35,571.05
XS GIS Cut Line= 4
  1056724.959209   683650.207418  1056930.182987   683268.173206
   1056967.70469   683235.401087  1057393.299083   682624.821638
#Sta/Elev= 30
       0 1517.33    16.5  1515.3   42.08  1509.8   86.36 1503.47  210.94 1482.76
  259.31 1476.81   291.8 1470.13  310.51  1470.4   327.7 1466.97  350.41 1464.09
  370.53 1460.25  386.85 1453.85  398.53 1450.76  415.32 1449.06  419.87 1447.23
  429.14  1441.1  435.29 1442.78   463.1 1446.69  477.71  1450.3  604.46 1448.88
  726.25  1448.7  888.69 1450.81 1002.73 1453.72 1063.62 1456.41 1103.79 1460.89
 1116.27 1460.98 1132.79 1465.41 1146.77 1466.55 1162.93 1470.24 1227.76 1491.07
#Mann= 3 , 0 , 0
       0     .08       0  415.32    .045       0  477.71     .07       0
Bank Sta=415.32,477.71
Exp/Cntr=0.3,0.1

Type RM Length L Ch R = 1 ,52905.23,485.45,471.01,456.72
XS GIS Cut Line= 5
  1056594.192878   684464.097187   1057109.71902   683894.805655
   1057393.48173   683445.201239  1057411.722254   683233.825543
   1057645.11599   682596.517269
#Sta/Elev= 30
       0  1509.4   75.48 1510.49  116.92 1514.01  239.66 1513.75  334.26 1521.05
     372 1517.23  419.51 1505.52  446.82 1513.09  546.21 1532.27  681.03 1566.35
  716.48 1567.45   759.6 1560.65  799.68    1550  855.17 1529.69  894.37  1512.5
  920.35 1498.15 1013.73 1483.26 1050.59 1460.37 1101.27  1462.2 1127.46 1451.83
 1151.39 1450.48 1337.76  1449.5  1366.7 1446.39 1398.22  1439.3 1427.74 1448.38
 1758.15 1448.61 1870.34 1452.99 1937.16 1476.74  2055.5 1502.56 2190.55 1564.06
#Mann= 3 , 0 , 0
       0     .07       0  1366.7    .045       0 1427.74     .07       0
Bank Sta=1366.7,1427.74
Exp/Cntr=0.3,0.1

Type RM Length L Ch R = 1 ,52434.23,469.16,466.12,451.25
XS GIS Cut Line= 3
  1058131.128366   684796.231566  1057769.567097   683051.877202
  1057753.406948   682458.266123
#Sta/Elev= 30
       0 1647.77   98.77 1637.62  181.47 1624.67  241.21 1606.92  254.91 1595.21
   268.1 1588.84   276.4 1589.86  312.88 1575.01   353.8 1564.53  416.17 1553.61
  457.78 1539.23  529.16 1529.06  649.67  1500.5  842.72 1460.52  862.95 1459.69
  871.21 1456.01 1144.34 1447.69 1690.73 1447.37 1714.74 1444.99 1743.53 1436.77
 1764.31 1446.18 1902.62 1449.01 1946.25 1454.54 2014.79 1478.61 2106.58 1498.65
 2152.99  1517.7 2237.34 1560.35 2258.61 1567.18 2327.89 1583.21 2375.26 1588.35
#Mann= 3 , 0 , 0
       0     .07       0 1714.74    .045       0 1764.31     .07       0
Bank Sta=1714.74,1764.31
Exp/Cntr=0.3,0.1

Type RM Length L Ch R = 1 ,51968.11,512.99,520.15,526.34
XS GIS Cut Line= 3
  1058522.545392    684156.49378  1058114.059373   682903.541551
  1057831.261392   682345.801095
#Sta/Elev= 30
       0 1510.47   58.11 1503.61  114.78 1494.38   159.2 1492.53  319.87 1471.81
  362.61 1469.67  371.09 1465.62  401.07 1465.65  422.59 1455.73  481.31 1451.44
  768.75 1445.58 1219.06  1446.8  1229.2 1438.93 1252.97 1436.15 1301.24 1446.34
 1338.79 1448.26 1351.45 1450.39 1390.86 1465.18 1441.71 1478.35 1475.53  1484.4
  1560.9 1492.69 1606.54 1500.32 1633.64 1509.46  1653.9 1513.84 1705.74 1536.18
 1837.49  1575.8 1853.98 1580.34 1887.55 1586.12 1905.79 1591.44  1943.2 1596.43
#Mann= 3 , 0 , 0
       0     .07       0 1219.06    .045       0 1301.24      .1       0
Bank Sta=1219.06,1301.24
Exp/Cntr=0.3,0.1

Type RM Length L Ch R = 1 ,51447.96,519.07,484.97,445.53
XS GIS Cut Line= 4
  1058523.349805    684592.19796  1058726.788363   683359.160561
  1058573.606115   682667.876561  1058390.176991   682244.184984
#Sta/Elev= 30
       0 1557.12   21.56 1552.99   85.57 1532.54  114.82 1528.41  184.04 1533.89
  237.88 1529.58  322.16 1519.76  407.65 1505.15  470.01 1503.04  570.44 1491.01
  753.05 1478.01   767.6 1471.51  809.29 1470.01  888.04  1460.8 1138.76 1461.67
 1178.18 1459.64 1229.48 1448.53 1294.99 1446.26 1772.83 1444.47 1817.67 1435.26
 1852.22 1444.52  2099.7 1445.91 2183.21 1451.21  2242.8 1463.87 2260.88 1469.97
 2289.13 1480.99 2312.04 1492.46 2323.17 1500.59 2343.79 1508.49 2419.45 1523.86
#Mann= 3 , 0 , 0
       0     .07       0 1772.83    .045       0 1852.22     .07       0
Bank Sta=1772.83,1852.22
Exp/Cntr=0.3,0.1

Type RM Length L Ch R = 1 ,50962.98,101.2,302.06,384.11
XS GIS Cut Line= 5
   1059851.19161   684553.334274  1059695.736981   683478.106256
  1059140.353568   682748.356446  1058456.362066   682141.941398
  1057579.084241   681676.562941
#Sta/Elev= 30
       0 1652.26  502.96 1542.26  666.22 1510.85   760.1 1498.82  854.35 1491.12
  941.55 1489.65 1001.12 1494.53 1086.41 1508.64  1153.7 1509.57 1305.16 1502.29
 1362.27 1493.64 1393.68 1495.65 1491.65 1485.89 1692.06 1477.67 1888.58 1453.87
 2070.82 1449.44 2170.43 1443.03 2202.57 1434.93 2223.35 1443.93 2685.03 1448.36
 2789.35 1473.01 2838.25 1492.71 2909.18 1503.02 3114.75 1508.78 3230.75  1505.1
 3273.61 1497.58 3315.49 1500.39 3398.76 1495.46 3602.05 1508.62 3910.64 1553.43
#Mann= 3 , 0 , 0
       0     .07       0 2170.43    .045       0 2223.35     .07       0
Bank Sta=2170.43,2223.35
Exp/Cntr=0.5,0.3

Type RM Length L Ch R = 1 ,50660.93,235.73,108.13,97.8
BEGIN DESCRIPTION:
Upstream xs of Bridge 37111-0245
END DESCRIPTION:
XS GIS Cut Line= 6
  1059763.114791   683474.897768  1059103.519032    682662.47853
  1059204.459083   682497.303873  1059301.728613   682308.270654
  1059311.124398   681954.339368  1058700.723014    680795.56904
#Sta/Elev= 30
       0  1517.8    89.5  1521.6   329.4  1497.8   615.1  1486.8   791.9    1472
   958.4  1448.1  1152.2  1444.5    1195    1437    1243  1431.6    1255  1434.5
  1385.8  1443.5    1547  1443.8    1601  1452.6  1738.2  1515.5  1956.8  1535.6
  2062.3  1520.1  2157.9  1484.9  2227.3  1480.6  2293.5  1530.6  2347.7  1561.3
  2405.1  1559.8  2487.3  1528.3  2546.6  1556.5    2620  1579.3  2683.4  1606.9
  2725.7  1625.9  2782.2    1661  2842.9  1684.5  2895.9  1688.3  3116.4  1659.5
#Mann= 3 , 0 , 0
       0     .07       0    1195    .045       0    1255     .07       0
#XS Ineff= 2 , 0
       0  1102.7  1446.3  1347.3       0  1446.9
Permanent Ineff=
       F       F
Bank Sta=1195,1255
Exp/Cntr=0.5,0.3

Type RM Length L Ch R = 3 ,50593.61,,,
BEGIN DESCRIPTION:
Bridge : 37111-0245, Lavender Rd. SR1129
END DESCRIPTION:
Bridge Culvert--1,0,-1,-1, 0
Deck Dist Width WeirC Skew NumUp NumDn MinLoCord MaxHiCord MaxSubmerge Is_Ogee
57.3,20,2.6,0, 84, 91, , , 0.95, 0, 0,0,,
    1017  1022.3  1026.7  1033.2  1035.8  1037.3  1039.8  1052.1  1058.2  1064.2
    1072  1074.1  1075.8  1091.9  1096.1  1108.6  1115.6  1121.3  1130.4  1131.5
  1132.3  1141.9  1147.9  1152.9    1160    1160    1290    1290    1290  1291.4
  1292.5  1292.9  1298.6  1308.7    1313  1319.2  1340.3  1349.5  1354.4  1365.5
  1365.9  1368.9  1376.5  1381.4  1382.6  1382.7  1383.1  1392.8  1396.6  1403.1
    1411  1412.9    1416  1421.3  1424.5  1430.5  1432.8  1437.1  1446.4  1447.2
  1448.4  1458.1  1464.6  1468.7    1476  1480.4  1486.2  1490.7    1498  1502.5
  1507.1  1511.4  1519.9  1522.9  1525.1  1532.5  1536.3  1544.6  1546.7  1554.8
  1559.5  1593.1  1597.7  1721.3
  1447.6  1447.5  1447.5  1447.6  1447.6  1447.6  1447.6  1447.4  1447.3  1447.1
  1446.9  1446.8  1446.8  1446.8  1446.8  1446.8  1446.8  1446.8  1446.6  1446.5
  1446.6  1446.6  1446.4  1446.4    1447    1447    1447    1447    1447    1447
    1447    1447    1447    1447    1447    1447    1447    1447    1447  1447.5
  1447.5  1447.5  1447.5  1447.5  1447.5  1447.5  1447.5  1447.5  1447.5  1447.5
  1447.5  1447.5  1447.5  1447.5  1447.5  1447.5  1447.5  1447.5  1447.5  1447.5
  1447.5  1447.5  1447.5  1447.5  1447.5  1447.6  1448.2  1448.4  1449.1  1449.4
  1449.6  1449.8  1450.2  1450.4  1450.5  1450.8    1451  1454.2  1454.1  1457.8
  1461.2  1478.8  1480.6  1511.3
                                                                                
                                                                                
                                          1444.6  1444.5
                                                                                
                                                                                
                                                                                
                                                                                
                                                                                
                                
   609.3   680.8   682.3   684.8   697.1   703.2   709.2     717   719.1   720.8
   736.9   741.1   753.6   760.6   766.3   775.4   776.5   777.3   786.9   792.9
   797.9     808   810.1   810.4   871.1     880     880    1010    1010  1010.5
  1010.9  1013.9  1021.5  1026.4  1027.6  1027.7  1028.1  1037.8  1041.6  1048.1
    1056  1057.9    1061  1066.3  1069.5  1075.5  1077.8  1082.1  1091.4  1092.2
  1093.4  1103.1  1109.6  1113.7    1121  1125.4  1131.2  1135.7    1143  1147.5
  1152.1  1156.4  1164.9  1167.9  1170.1  1177.5  1181.3  1189.6  1191.7  1199.8
  1204.5  1238.1  1242.7  1252.4    1282  1288.1  1296.3  1313.7    1335  1345.4
    1355  1355.8  1373.5  1373.8  1401.2  1423.3  1427.2  1429.1  1433.4  1442.4
  1452.5
  1447.7  1447.6  1447.6  1447.6  1447.4  1447.3  1447.1  1446.9  1446.8  1446.8
  1446.8  1446.8  1446.8  1446.8  1446.8  1446.6  1446.5  1446.6  1446.6  1446.4
  1446.4  1446.5  1446.5  1446.5  1446.4    1447    1447    1447    1447  1447.1
  1447.3  1447.4  1447.5  1447.5  1447.5  1447.5  1447.5  1447.5  1447.5  1447.5
  1447.5  1447.5  1447.5  1447.5  1447.5  1447.5  1447.5  1447.5  1447.5  1447.5
  1447.5  1447.5  1447.5  1447.5  1447.5  1447.6  1448.2  1448.4  1449.1  1449.4
  1449.6  1449.8  1450.2  1450.4  1450.5  1450.8    1451  1454.2  1454.1  1457.8
  1461.2  1478.8  1480.6  1486.2    1501  1503.7  1507.7  1512.2  1518.9  1522.4
  1525.2  1525.4  1530.2  1530.2  1536.6  1543.7  1545.1  1545.5    1545  1545.4
    1544
                                                                                
                                                                                
                                                  1444.6  1444.5
                                                                                
                                                                                
                                                                                
                                                                                
                                                                                
                                                                                
        
Pier Skew, UpSta & Num, DnSta & Num=  ,1195, 2 ,915, 2 , 0 , 0 , 0 ,,
       1       1
    1436  1445.1
       1       1
    1436  1445.1
Pier Skew, UpSta & Num, DnSta & Num=  ,1230, 2 ,950, 2 , 0 , 0 , 0 ,,
       1       1
  1432.4  1445.1
       1       1
  1432.4  1445.1
Pier Skew, UpSta & Num, DnSta & Num=  ,1265, 2 ,985, 2 , 0 , 0 , 0 ,,
       1       1
    1434  1445.1
       1       1
    1434  1445.1
BR Coef=-1 , 1 , 1 ,2.5, 0 ,,,0.8,0,1.2,0,
WSPro=,,,, 1 ,,,, 0 ,,,, 0 ,,,,-1 ,-1 ,-1 , 0 , 0 , 0 , 0 , 0
BC Design=,, 0 ,, 0 ,,,,,,

Type RM Length L Ch R = 1 ,50552.79,78.13,79.96,82.1
BEGIN DESCRIPTION:
Down stream xs of Bridge 37111-0245
END DESCRIPTION:
XS GIS Cut Line= 6
  1059646.368465   683194.706548  1059201.706183    682660.64325
  1059368.624583   682374.339025  1059391.312041    682315.35161
  1059406.043642    681958.25514  1059408.419521   681900.663186
#Sta/Elev= 30
       0  1503.4    43.5  1499.4    68.8  1501.1   100.6  1497.2   196.7  1496.3
   224.3  1491.7   261.1  1490.7   272.7  1487.5   310.6  1486.7   317.6  1484.7
   408.7  1478.8   477.6  1469.1   539.6  1455.5     613  1447.2   723.4  1443.2
   865.5  1444.5     909  1439.2     963  1431.6     985    1435  993.071439.681
    1008  1444.4  1035.9  1446.5  1171.9    1450  1231.3  1461.9  1318.9  1509.9
  1344.6  1516.3  1409.7    1540  1429.7  1544.9  1460.4  1557.2  1504.6  1568.3
#Mann= 3 , 0 , 0
       0     .07       0     909    .045       0  993.07      .1       0
#XS Ineff= 2 , 0
       0   849.2  1446.3  1040.8       0  1447.4
Permanent Ineff=
       F       F
Bank Sta=909,993.07
Exp/Cntr=0.5,0.3

Type RM Length L Ch R = 1 ,50472.84,420.74,392.12,361.6
XS GIS Cut Line= 6
  1059710.578954   683229.730426  1059276.339091   682664.018228
  1059441.367063   682401.082415   1059467.33874   682333.556095
  1059482.307552   681970.709428   1059484.68347   681913.117473
#Sta/Elev= 30
       0 1503.11   95.82 1498.96  118.36 1500.46  200.28 1490.61  251.12 1491.64
  332.67 1486.26  455.55  1472.4   512.7 1464.33  568.93 1453.06  597.53 1449.08
  734.52 1442.57  952.46  1443.7  960.91 1435.62  968.58 1433.52  990.25 1439.13
 1003.08 1444.28  1075.6 1442.29 1111.79 1445.07 1141.22 1453.68 1190.44 1484.04
 1204.94 1487.36 1222.03 1488.48 1239.79 1487.46 1280.74 1477.39 1306.54    1479
 1349.91 1494.26 1391.91 1511.42  1470.3 1550.34 1506.59 1571.49 1516.74 1576.03
#Mann= 3 , 0 , 0
       0     .07       0  952.46    .045       0 1003.08      .1       0
Bank Sta=952.46,1003.08
Exp/Cntr=0.3,0.1

Type RM Length L Ch R = 1 ,50080.71,521.75,523.37,527.83
XS GIS Cut Line= 3
  1059792.301402   683276.428995  1059790.964428   682413.078979
  1059739.765526   681898.822041
#Sta/Elev= 30
       0 1506.72   34.05 1501.89   48.97 1498.24   96.95 1496.31  111.54 1488.52
  130.36 1482.13  230.34 1458.52  276.74 1451.32  312.65 1447.86  341.02 1445.48
  455.78 1441.55  745.08 1442.87  775.62 1433.22  789.25 1433.96  819.43 1443.44
  832.43 1446.75  842.52  1455.1  872.87 1469.04  911.59 1480.63     946 1487.73
  987.62 1499.33 1018.03 1517.12  1027.4 1517.33 1081.49 1537.68 1122.18 1550.76
 1189.45 1560.68 1224.88 1569.38 1292.09 1588.65 1347.85 1601.12 1380.15 1606.41
#Mann= 3 , 0 , 0
       0     .07       0  745.08    .045       0  819.43      .1       0
Bank Sta=745.08,819.43
Exp/Cntr=0.3,0.1

Type RM Length L Ch R = 1 ,49557.34,834.12,827.24,810.18
XS GIS Cut Line= 3
  1060211.156984   684040.163195  1060216.360407   682689.163821
  1060294.310699   681863.798163
#Sta/Elev= 30
       0 1533.29   166.7 1528.07  207.76 1529.41  267.99 1537.12  318.33 1535.87
  391.58 1527.22  453.09 1516.33   511.7 1501.76  551.44 1500.29   560.5 1495.19
  692.08 1466.23  756.53 1455.07  819.92 1448.51 1077.47 1440.56 1291.76 1440.91
 1319.56 1431.96 1351.01  1440.6 1375.82 1443.14 1384.49 1441.41 1434.63  1466.6
 1499.77 1481.61 1572.74 1493.31 1620.44 1496.57 1728.68 1488.73 1775.06 1491.48
 1837.88 1501.25 2006.04 1540.32 2065.71  1546.8 2124.65 1564.54 2180.05 1577.38
#Mann= 3 , 0 , 0
       0     .07       0 1291.76    .045       0 1351.01      .1       0
Bank Sta=1291.76,1351.01
Exp/Cntr=0.3,0.1

Type RM Length L Ch R = 1 ,48730.1 ,532.3,541.38,545.72
XS GIS Cut Line= 3
   1061249.14424   684024.949754  1060979.542551   682390.255556
  1060965.400483    682060.27402
#Sta/Elev= 30
       0 1494.33  128.72 1488.96  149.19  1496.7  173.26 1501.73  339.22 1508.46
  392.14 1502.68  521.17 1480.98  650.62 1447.56  704.63 1443.74  811.44 1441.85
  822.99 1443.75  994.52 1439.07  1453.6 1440.43 1473.49 1438.21 1502.53  1430.5
  1514.2 1437.47 1552.51 1440.39 1567.78 1444.67 1584.18 1452.72 1606.79 1468.69
 1619.69 1471.38 1636.95 1487.32 1662.53  1501.7 1698.87  1514.8 1741.73 1537.38
 1830.57 1574.21 1877.93  1583.7 1898.04 1584.46 1946.88 1575.97 1987.06 1582.76
#Mann= 3 , 0 , 0
       0     .07       0 1473.49    .045       0  1514.2      .1       0
Bank Sta=1473.49,1514.2
Exp/Cntr=0.3,0.1

Type RM Length L Ch R = 1 ,48188.72,580.26,600,635.71
XS GIS Cut Line= 3
  1061474.514854   683856.316349  1061523.326149   682472.800009
  1061500.273165   681931.850479
#Sta/Elev= 30
       0 1529.51   57.72 1539.25  127.87 1538.64  166.42 1545.83  191.43 1546.06
  279.11 1535.41  317.48 1527.59  382.11 1523.97  404.28 1520.72  465.73 1499.35
  549.66 1480.13  693.77 1458.16  734.79 1443.15  764.42 1440.63  828.17  1438.4
 1103.97 1437.31 1254.47 1440.47 1352.16 1439.16 1367.24 1433.29 1384.38    1430
 1415.57 1437.73 1493.89 1442.07 1586.26 1487.86 1661.12 1529.67 1687.85 1540.94
 1723.79 1546.23 1789.68 1541.39 1846.01 1542.59 1906.01 1553.33 1925.82 1553.95
#Mann= 3 , 0 , 0
       0     .07       0 1352.16    .045       0 1415.57      .1       0
Bank Sta=1352.16,1415.57
Exp/Cntr=0.3,0.1

Type RM Length L Ch R = 1 ,47588.72,579.24,591.57,585.1
XS GIS Cut Line= 3
  1061525.984678   684011.930983  1061990.503962    682743.58892
  1062341.420475   682321.769712
#Sta/Elev= 30
       0 1514.44   39.31 1522.35   250.7 1538.49  307.15 1546.48   363.8 1544.74
  465.57  1523.7  533.87 1499.87  569.27 1492.67  603.74 1482.63  667.93 1473.58
  774.23 1447.63  811.41 1443.04  893.98 1438.14   998.2  1436.3 1268.13 1436.85
 1330.15 1439.56 1350.73 1428.35 1384.13 1436.64 1482.02 1438.71 1506.56 1447.44
  1533.8 1463.01 1568.47 1471.36 1582.24 1478.95 1626.44 1492.87 1681.15 1519.75
 1747.68 1545.81 1779.37 1563.77 1834.26 1580.37 1876.18 1587.52 1899.43 1588.98
#Mann= 3 , 0 , 0
       0     .07       0 1330.15    .045       0 1384.13      .1       0
Bank Sta=1330.15,1384.13
Exp/Cntr=0.3,0.1

Type RM Length L Ch R = 1 ,46997.15,595.98,547.07,494.3
XS GIS Cut Line= 3
  1061548.524986   684438.846931  1062377.910418   683076.285102
  1062366.417519   682509.488987
#Sta/Elev= 30
       0 1540.49  162.89 1535.97  249.83  1526.8  302.82 1518.22  317.77 1514.74
  353.75 1500.23  395.62 1497.36  423.96 1499.19  478.22 1492.45  579.64 1493.81
  704.47 1506.54  747.45 1514.85   826.9 1518.71  930.84 1494.98 1119.88 1443.14
  1238.4 1436.77 1402.62 1436.12 1429.84 1428.04 1442.54 1427.84 1466.82 1434.89
 1498.82 1438.16 1663.72 1436.97 1776.39  1500.2 1795.97 1509.34 1845.06 1524.48
 1991.81 1549.59 2088.08 1556.85 2104.22 1560.01 2119.97  1567.7 2162.05 1571.13
#Mann= 3 , 0 , 0
       0     .07       0 1402.62    .045       0 1466.82     .07       0
Bank Sta=1402.62,1466.82
Exp/Cntr=0.3,0.1

Type RM Length L Ch R = 1 ,46450.07,793.02,839.64,853.37
XS GIS Cut Line= 4
  1063156.940353   684540.298532  1062839.404211   683213.281801
  1062544.532576   682555.491302  1062518.609756   681869.233011
#Sta/Elev= 30
       0 1561.63  194.08 1530.58  254.36 1527.47     276 1520.89  322.81 1521.26
  411.46 1513.24  719.51 1532.18   878.5 1530.05  986.42 1502.56 1071.48 1471.39
 1176.53 1437.89 1291.89 1433.51 1466.49 1435.79 1510.19 1426.06 1546.18 1436.34
  1827.3 1437.05 1923.94 1485.13 1958.48 1496.91 2011.92 1509.51 2074.95 1530.86
 2181.94 1542.38 2235.48 1544.08 2366.87 1582.05 2438.68  1582.8 2498.54 1574.65
  2531.1 1563.88 2563.72 1557.95 2612.19 1568.41 2678.54 1573.78 2772.09 1567.19
#Mann= 3 , 0 , 0
       0      .1       0 1466.49    .045       0 1546.18     .07       0
Bank Sta=1466.49,1546.18
Exp/Cntr=0.3,0.1

Type RM Length L Ch R = 1 ,45610.44,395.72,421.72,440.06
XS GIS Cut Line= 3
  1063170.269774   683794.592151  1063443.463963   682974.593727
  1064438.858757   681686.182306
#Sta/Elev= 30
       0  1557.2    78.2 1536.66  117.86 1517.99  191.68 1502.42  248.91 1499.49
  278.11  1509.8  330.14 1512.95  416.24 1490.81  525.58 1469.94  594.19 1444.76
  628.21 1438.17  710.28  1432.6  820.88 1433.74  838.42 1424.85  875.81  1432.5
  909.91  1438.8  920.85 1448.85  991.74 1476.13 1063.77 1493.15 1130.33 1500.71
 1288.43 1503.92 1474.97 1492.15 1581.61  1481.1  1704.8 1487.26 1983.88 1478.98
  2118.1 1496.53 2257.92 1527.63 2326.13 1537.72 2377.99 1535.97 2492.44 1519.75
#Mann= 3 , 0 , 0
       0      .1       0  820.88    .045       0  875.81      .1       0
Bank Sta=820.88,875.81
Exp/Cntr=0.3,0.1

Type RM Length L Ch R = 1 ,45188.72,473.65,497.27,509.44
XS GIS Cut Line= 3
  1063322.113184   683839.073137  1063690.522781   683313.835898
  1064088.270605   682920.698975
#Sta/Elev= 30
       0 1581.44    49.5 1564.96   71.18 1545.72  114.64  1532.9     199 1540.84
  208.48 1539.26   228.4 1546.56   279.5 1557.66  315.17 1554.71  355.25 1543.61
  378.33 1529.01  406.19 1517.45  451.76 1505.08  485.04  1492.7  570.33 1455.25
  609.05 1442.34  624.52 1433.04  641.83 1423.67  687.06 1432.73  745.66 1432.97
  770.14 1441.44  780.19 1441.68  818.16 1464.49  837.72 1470.03   851.4 1479.53
  895.61 1498.36  963.38  1535.2 1069.11 1563.83  1138.9  1565.4 1200.81 1553.66
#Mann= 3 , 0 , 0
       0      .1       0  624.52    .045       0  687.06      .1       0
Bank Sta=624.52,687.06
Exp/Cntr=0.3,0.1

Type RM Length L Ch R = 1 ,44691.45,434.33,462.86,486.33
XS GIS Cut Line= 3
  1063697.581057   683691.930299  1064240.487308   683392.570797
  1064514.477405   683204.836841
#Sta/Elev= 30
       0 1565.55   14.79 1561.93    39.5 1547.74   67.51 1537.99  104.35 1530.46
  140.26 1514.79  191.19 1486.72  250.85 1476.62  270.17 1471.09  340.76  1437.6
  372.47 1432.24  387.86 1431.47  462.71 1432.35  493.42  1430.8  531.01 1422.86
  568.35 1427.54  580.51 1431.51  613.24 1431.72  630.47 1435.97  649.24 1447.83
  662.25 1451.85  673.51 1463.74  708.52 1484.15   765.4 1513.95  802.73 1526.61
  842.24 1545.14  884.49 1547.96   917.4 1536.51  927.32 1534.43  952.11 1533.42
#Mann= 3 , 0 , 0
       0      .1       0  493.42    .045       0  580.51      .1       0
Bank Sta=493.42,580.51
Exp/Cntr=0.3,0.1

Type RM Length L Ch R = 1 ,44228.59,842.7,839.87,840.04
XS GIS Cut Line= 3
  1063814.280547   683783.260344  1064306.447909   683752.816996
  1064925.462492   683752.816996
#Sta/Elev= 30
       0 1526.37    38.2 1516.67  115.39 1504.79   241.5  1473.1  274.69 1460.46
   315.8 1458.28  364.98 1445.69  391.09 1441.63   420.9 1438.08  508.83 1436.15
  556.55 1432.36  614.49 1432.25  643.14 1428.74  663.54 1422.52  682.97 1428.89
  702.45 1434.98  708.96 1441.12  722.28 1448.65  742.06 1456.06   853.4 1507.43
  881.56 1517.06  893.87 1517.52  922.37 1523.51  940.53  1530.7   951.9 1532.75
  963.79 1542.01 1006.92 1562.63 1056.06 1577.43 1078.99  1578.7 1112.12 1572.77
#Mann= 3 , 0 , 0
       0      .1       0  643.14    .045       0  682.97      .1       0
Bank Sta=643.14,682.97
Exp/Cntr=0.3,0.1

Type RM Length L Ch R = 1 ,43388.72,645.43,596.65,540.63
XS GIS Cut Line= 4
  1063301.817606   684244.984358  1063851.275127    684203.58238
  1064481.504541   684226.054142  1064751.912119   684015.786636
#Sta/Elev= 30
       0 1539.81  140.15 1534.64  227.82 1527.13  256.35 1531.23  305.17 1518.48
  386.34 1509.47  426.72 1500.22   469.6 1482.52  477.46 1478.17  496.87  1451.4
  508.58 1451.54  545.43 1427.28  551.01 1419.71  579.64 1426.11  604.99 1428.14
  759.88 1427.46  862.12 1435.58  892.96 1443.36  966.92 1450.45  988.94 1459.87
  1009.8 1462.86  1017.5 1466.62 1135.75 1488.37 1177.91 1493.64 1209.53 1489.29
 1345.75 1489.63 1466.69  1515.6 1482.65  1515.3  1497.5 1527.51 1524.18 1537.84
#Mann= 3 , 0 , 0
       0      .1       0  545.43    .045       0  579.64     .07       0
Bank Sta=545.43,579.64
Exp/Cntr=0.3,0.1

Type RM Length L Ch R = 1 ,42792.07,50.67,50.67,50.67
XS GIS Cut Line= 4
  1063970.040233   684824.406766   1064241.54435   684650.459217
  1064318.530185   684515.417491  1064632.292656   684231.652024
#Sta/Elev= 30
       0 1563.45   79.78 1546.31  125.73 1532.67  161.68 1518.66   278.6 1463.22
  296.34 1443.09  298.34 1442.06  311.82 1439.27  333.82 1439.08  361.96 1434.23
  376.71 1426.93  381.12 1423.08  390.78 1418.84  403.15 1418.99  433.99 1424.81
  463.93 1425.71  480.16 1428.28  500.56 1433.95  567.29 1436.92   595.2 1443.75
  627.81 1445.18  643.06 1449.19  693.67 1470.58  711.37 1474.61  724.74 1480.59
  750.36 1486.16  774.58  1495.3  828.48 1498.67  883.49 1497.38  900.94 1500.15
#Mann= 3 , 0 , 0
       0      .1       0  376.71    .045       0  433.99      .1       0
Bank Sta=376.71,433.99
Exp/Cntr=0.5,0.3

Type RM Length L Ch R = 1 ,42741.4 ,55.74,55.74,57.28
BEGIN DESCRIPTION:
Upstream xs of Bridge 37111-0239
END DESCRIPTION:
XS GIS Cut Line= 4
  1063997.013261   684866.507329  1064278.883989    684685.91806
  1064358.546451   684546.181199  1064632.292656   684264.364646
#Sta/Elev= 30
       0  1564.1    96.8    1540   115.7  1533.7   159.1  1518.5   194.8  1503.5
   280.1  1463.7   311.9  1450.6   328.3    1442   340.7  1437.7   368.6  1436.9
   382.3  1434.3     392  1429.4     410  1421.5     415  1420.7     420  1416.4
     428  1414.9     448  1415.2     465  1421.4     493  1428.5   495.6  1431.6
   506.3  1434.6   565.9  1434.7   596.7  1440.6   648.2  1446.1   660.3  1449.9
     710  1473.4   780.3  1491.5   820.1  1498.7     851  1501.3   888.5  1499.2
#Mann= 3 , 0 , 0
       0      .1       0     392    .045       0     493      .1       0
#XS Ineff= 2 , 0
       0   372.6  1436.1   512.4       0  1435.3
Permanent Ineff=
       F       F
Bank Sta=392,493
Exp/Cntr=0.5,0.3
